--- MFReedyCrk.prj (project) ---

Proj Title=MFReedyCrk
Current Plan=p01
Default Exp/Contr=0,0
English Units
Geom File=g01
Flow File=f01
Plan File=p01
BEGIN DESCRIPTION:
AMEC Environment & Infrastructure, 2013
Projection: NAD 1983 State Plane West Virginia South FIPS 4702 (US Feet)
Vertical Datum: NAVD 1988
END DESCRIPTION:
DSS Export Rating Curves= 0
DSS Export Rating Curve Sorted= 0
DSS Export Volume Flow Curves= 0
DXF Filename=.\Hec_working\MFReedyCrk.
DXF OffsetX= 0
DXF OffsetY= 0
DXF ScaleX= 0
DXF ScaleY= 0

--- MFReedyCrk.p01 (plan) ---

Plan Title=Floodplain
Program Version=4.00
Geom File=g01
Flow File=f01
K Sum by GR=0
Std Step Tol=0.01
Critical Tol=0.01
Num of Std Step Trials=20
Max Error Tol=0.3
Flow Tol Ratio=0.001
Split Flow NTrial=30
Split Flow Tol=0.02
Split Flow Ratio=0.02
Log Output Level=0
Friction Slope Method=1
Unsteady Friction Slope Method=2
Unsteady Bridges Friction Slope Method=1
Global Log Level=0
CheckData=False
Run HTab=0
Run UNet=0
Run PostProcess=0
UNET Theta=0
UNET Theta Warmup=0
UNET ZTol=0
UNET ZSATol=0
UNET MxIter=0
UNET MaxInSteps=0
UNET DtIC=0
UNET DtMin=0
UNET MaxCRTS=0
UNET WFStab=0
UNET SFStab=0
UNET WFX=0
UNET SFX=0
UNET DSS MLevel=0
UNET DZMax Abort=0
UNET Convert EG Bridges=0
UNET Use Existing IB Tables=0
UNET Froude Limit=0
UNET Froude Power=0
Write IC File=0
Echo Input=False
Echo Output=False
Write Detailed=0

--- MFReedyCrk.f01 (steady flow) ---

Flow Title=NFF Regression Equation
Program Version=4.10
Number of Profiles= 1
Profile Names=P100yr
River Rch & RM=MFReedyCrk,Main            ,57747.1
888.6882
River Rch & RM=MFReedyCrk,Main            ,57040.6
894.6682
River Rch & RM=MFReedyCrk,Main            ,56284.2
987.8857
River Rch & RM=MFReedyCrk,Main            ,53593
1074.293
River Rch & RM=MFReedyCrk,Main            ,52290.1
1178.452
River Rch & RM=MFReedyCrk,Main            ,51188.9
1295.857
River Rch & RM=MFReedyCrk,Main            ,49189
1427.435
River Rch & RM=MFReedyCrk,Main            ,47184.8
1557.952
River Rch & RM=MFReedyCrk,Main            ,46743.2
1614.526
River Rch & RM=MFReedyCrk,Main            ,45017.4
1772.399
River Rch & RM=MFReedyCrk,Main            ,37087.1
1919.612
River Rch & RM=MFReedyCrk,Main            ,36224.7
2252.696
River Rch & RM=MFReedyCrk,Main            ,35894.8
2395.672
River Rch & RM=MFReedyCrk,Main            ,32015.6
2540.042
River Rch & RM=MFReedyCrk,Main            ,25244.8
 2734.71
River Rch & RM=MFReedyCrk,Main            ,22486.3
3037.982
River Rch & RM=MFReedyCrk,Main            ,19055.3
3320.918
River Rch & RM=MFReedyCrk,Main            ,12787.6
3630.632
River Rch & RM=MFReedyCrk,Main            ,514.9
4033.903
River Rch & RM=MFReedyCrk,Main            ,13.9
4038.224
Boundary for River Rch & Prof#=MFReedyCrk,Main            , 1
Up Type= 0
Dn Type= 1
Dn Known WS=680
DSS Import GetInterval= 0
DSS Import GetPeak= 0
DSS Import FillOption= 0

--- MFReedyCrk.g01 (geometry) ---

Geom Title=USGS 3m DEM
Program Version=4.10

River Reach=MFReedyCrk      ,Main
Reach XY= 30
     1831130.473      650451.321     1831540.162      653056.453
     1831085.014      654807.052     1832877.201      656635.965
      1832797.21      658064.205     1833667.226      659367.917
      1835091.29      660314.543     1835504.564      661337.516
     1835571.225      664768.654     1836914.429      666652.069
     1836362.556      668142.858     1837279.198      669141.434
     1838498.143      669547.351     1838386.959      669983.269
     1839380.322      670856.928     1839593.893      671563.804
     1838841.713      673849.325     1840455.015      675914.451
     1840037.153       676934.48     1841995.304      678995.583
     1842050.766      680588.203      1843113.66      680697.696
     1844185.152      682022.929     1844819.097      681701.671
     1845541.516      682792.415     1845482.383      683957.786
     1844733.808      685015.528     1847059.131      687379.347
     1846895.758      688996.276     1847963.768      690522.983

Type RM Length L Ch R = 1 ,57747.1 ,311.3,312.7,312.6
XS GIS Cut Line= 3
     1830779.767      650605.337     1831132.642      650461.083
      1831492.15      650333.765
#Sta/Elev= 30
       0  866.46    19.6  857.15    29.3  853.37    39.1  850.42   195.5   813.7
     215  809.44   234.6   805.8   254.2  802.64   273.7  800.25   293.2  798.32
   322.6  796.43   373.7  794.94   381.2  794.69   388.7  795.75     391  796.08
   400.8   799.6   420.3  807.46   547.5  850.81   557.2  854.23     567  858.15
   576.8  863.58   615.9  892.06   625.7  898.92   635.5   904.4   664.8  916.93
   674.6  920.66   713.7  933.69   723.5   935.9   733.3  937.28   762.6  940.57
#Mann= 3 , 0 , 0
       0     .06       0   373.7    .045       0   388.7      .1       0
Bank Sta=373.7,388.7
XS Rating Curve= 0 ,0
Exp/Cntr=0.3,0.1

Type RM Length L Ch R = 1 ,57434.5 ,389.9,393.9,398.7
XS GIS Cut Line= 3
     1830886.578      650863.276     1831386.578      650693.832
     1831489.356      650582.721
#Sta/Elev= 30
       0  850.14     9.8  847.35    19.6  844.96    68.4     834    97.8  827.65
   166.2  814.69   195.5  809.87   205.3  808.66   215.1  807.78   371.5  795.95
     404  793.05   410.6  792.69     419  793.33   420.4  793.44   430.2  795.86
   449.7  802.24     479  811.09   537.4  827.26   556.3  833.34   575.2  840.08
   584.7  844.23   594.2  849.55   603.6   857.3   613.1  866.73   622.5  877.23
     632  886.36   641.4  892.79   650.9   897.7   669.8  904.18   679.3   906.8
#Mann= 3 , 0 , 0
       0     .06       0     404    .045       0     419      .1       0
Bank Sta=404,419
XS Rating Curve= 0 ,0
Exp/Cntr=0.3,0.1

Type RM Length L Ch R = 1 ,57040.6 ,305.5,305.1,303.9
XS GIS Cut Line= 4
     1830992.134      651177.165     1831187.114      651116.628
     1831474.181      651070.746     1831781.023      651082.721
#Sta/Elev= 30
       0  868.82    29.2  861.12    48.6   855.3    77.8  845.26   136.1  822.76
   165.3  812.24   194.4  803.12   204.2  800.48   213.8  798.55   233.2  796.91
   310.8   792.9   339.8  791.86   407.7  790.76   465.8  788.83   468.9   788.9
   475.5  789.05   483.9  790.83   494.9  795.62   514.1  804.89   523.7  808.36
     562  819.94     610   837.3   638.8  846.14   648.4  850.45   667.6  860.74
   696.4  878.17     706  883.36   715.6  887.04     754  898.04     802  910.35
#Mann= 3 , 0 , 0
       0     .06       0   468.9    .045       0   483.9     .07       0
Bank Sta=468.9,483.9
XS Rating Curve= 0 ,0
Exp/Cntr=0.3,0.1

Type RM Length L Ch R = 1 ,56735.5 ,442.6,451.3,456.7
XS GIS Cut Line= 3
     1830928.245      651385.498     1831214.356      651404.943
       1831708.8      651327.165
#Sta/Elev= 30
       0  898.31    38.2  890.97    47.8  888.53    57.4  885.42    76.5  877.96
    95.6   869.8   105.2  865.26   133.8  850.34   152.9  841.23   172.1  833.55
   191.2  826.79   210.3  820.98   296.6  797.25   306.4  795.05   316.2  793.92
     326  793.46   521.3  787.58   522.3  787.56   532.1  788.41   536.3  789.72
   541.9  791.47   561.6  801.12   571.4  804.79   581.2  807.57   600.8  811.81
   659.7  823.08     699  833.21   718.6  840.02   767.7  861.73   787.3  868.59
#Mann= 3 , 0 , 0
       0     .06       0   521.3    .045       0   536.3     .08       0
Bank Sta=521.3,536.3
XS Rating Curve= 0 ,0
Exp/Cntr=0.3,0.1

Type RM Length L Ch R = 1 ,56284.2 ,709.6,704.2,698.1
XS GIS Cut Line= 3
     1831072.229      651811.998     1831468.133      651791.818
     1831859.393      651843.484
#Sta/Elev= 30
       0  827.74    19.3  826.42      29  824.97    38.7  822.93     145  796.98
   154.7  794.97   164.4  793.64   366.2  784.81   367.4  784.79   381.2  785.22
     406   787.8   415.7  789.38   425.3  791.91   434.9  795.35   463.8  807.25
   492.7  820.17   531.2  839.09   540.8  844.68   550.4   851.4   569.7  866.13
   579.3  871.79   588.9  875.87   598.6  879.26   617.8  885.16   637.1  890.18
   656.3  893.67     743   905.9   752.6  906.77   771.8  907.54   791.1  907.17
#Mann= 3 , 0 , 0
       0     .06       0   366.2    .045       0   381.2     .08       0
Bank Sta=366.2,381.2
XS Rating Curve= 0 ,0
Exp/Cntr=0.3,0.1

Type RM Length L Ch R = 1 ,55580   ,330.2,330.6,332.6
XS GIS Cut Line= 3
     1831074.953      652482.721     1831466.642      652468.103
     1831740.107      652431.556
#Sta/Elev= 30
       0  845.08     9.8  842.04    19.6  839.27    29.4  836.72      98  819.59
     196  794.44   205.8  792.39   215.6  791.49   235.2  791.05     245  790.59
   303.8  787.33   352.8  784.47   384.5  782.28     392  782.04   399.5  782.48
   401.5   782.6     411  784.39   420.5   787.2     430  790.55   439.5  794.32
     449  798.56   458.6  803.19   487.1  818.08   496.6   822.8   506.1  827.28
   591.8  865.34   610.8   873.9   620.3   877.8   629.8  881.11   667.9  892.76
#Mann= 3 , 0 , 0
       0     .06       0   384.5    .045       0   399.5      .1       0
Bank Sta=384.5,399.5
XS Rating Curve= 0 ,0
Exp/Cntr=0.3,0.1

Type RM Length L Ch R = 1 ,55249.4 ,558.1,566.7,570.7
XS GIS Cut Line= 3
     1830942.134      653002.165     1831256.023      652802.165
     1831728.245      652782.721
#Sta/Elev= 30
       0  879.37    19.6  877.08    78.4  867.87      98  862.94   117.5  855.98
   137.1  843.95   146.9  838.89   156.7  835.14   176.3  828.87   195.9  823.49
   215.5   818.9   235.1  815.05   264.4  810.43     284  808.59   313.4  808.86
     333   807.9   352.6  804.76   401.1     795   430.1  790.82     459  788.26
   562.8  780.71   574.7  780.29   577.8  780.34     623  781.73   632.6  782.81
   642.3  785.19   719.4  812.72   767.6  829.26   806.2  841.52   844.8  852.69
#Mann= 3 , 0 , 0
       0     .06       0   562.8    .045       0   577.8     .08       0
Bank Sta=562.8,577.8
XS Rating Curve= 0 ,0
Exp/Cntr=0.3,0.1

Type RM Length L Ch R = 1 ,54682.7 ,422.6,418.6,419.4
XS GIS Cut Line= 3
     1831071.018      653163.618     1831435.526      653282.789
     1831807.015      653352.537
#Sta/Elev= 30
       0  840.92     9.8  837.82    39.3  828.99    68.8  820.81    98.3  813.02
   147.5  800.23   186.8  789.46   196.7   786.9   206.5  784.63   216.3  782.78
   226.2  781.62     236  781.16   324.5  778.99     376  777.91   383.5  777.85
     391  777.93   402.9  778.22   412.6  778.64   480.4  782.13   528.9  784.24
   538.6  785.53   548.3  787.96   596.7  802.54   664.6  824.51   674.2  827.71
   693.6  834.44   703.3  837.99     713  841.66   742.1  852.95   761.5  860.22
#Mann= 3 , 0 , 0
       0     .06       0     376    .045       0     391     .06       0
Bank Sta=376,391
XS Rating Curve= 0 ,0
Exp/Cntr=0.3,0.1

Type RM Length L Ch R = 1 ,54264.1 ,670.1,671.1,666.7
XS GIS Cut Line= 3
     1830956.879        653557.2     1831268.011      653586.698
     1831712.556      653698.889
#Sta/Elev= 30
       0  874.87    29.3  858.01    48.8  847.51    68.4  838.21    78.1     834
    97.7  827.14     127  819.02   156.3  812.28   185.6  806.52   234.4  798.24
   253.9   794.3   273.5  789.22     305  778.44   312.5  776.72     320  776.31
   322.3  776.19   458.8  781.68   507.6  783.19   517.4  783.62   527.1  784.98
   546.6  789.93   575.9  795.21   624.7  804.94   634.4  807.48     654  813.68
   702.7  831.03   722.2  839.09     732  843.79   741.8  849.19     771   867.5
#Mann= 3 , 0 , 0
       0      .1       0     305    .045       0     320     .06       0
Bank Sta=305,320
XS Rating Curve= 0 ,0
Exp/Cntr=0.3,0.1

Type RM Length L Ch R = 1 ,53593   ,402.6,408.5,413.3
XS GIS Cut Line= 4
     1830811.578      654310.498     1831178.245      654157.721
       1831483.8      654191.054     1831767.134      654085.498
#Sta/Elev= 30
       0  910.25    29.1  903.94    48.4  898.69   106.6  881.46     155  865.69
   174.4  858.42   222.8  838.47     310  803.92   339.1   793.5   358.5   788.1
   397.2  780.74   416.4  778.53   582.9     772   589.3  771.92   597.9  771.93
   608.5  772.01   618.1  772.72   627.8   774.8   685.4  795.17   733.8  808.81
   772.9  819.26   782.6   822.7   792.4  826.83   821.6  841.58   850.9  854.61
   928.9     885   948.4  891.46   967.9  897.24   987.4  901.91    1007  905.26
#Mann= 3 , 0 , 0
       0     .06       0   582.9    .045       0   597.9      .1       0
Bank Sta=582.9,597.9
XS Rating Curve= 0 ,0
Exp/Cntr=0.3,0.1

Type RM Length L Ch R = 1 ,53184.6 ,910.1,894.5,880.5
XS GIS Cut Line= 3
     1830901.777        654403.4     1831267.808      654552.961
      1831661.39      654690.715
#Sta/Elev= 30
       0  870.62    57.9  842.54    77.2  834.03    96.4  826.27   154.3  805.72
   241.1  778.18   250.8  775.62   260.4  773.87     270  772.92   390.6  769.09
   395.4  769.02   405.6  769.35   414.8  770.18   424.5  771.67   434.2  774.81
   453.6  786.32   463.3  789.44   511.8  800.98   589.4  816.35   608.8  819.74
   618.4  821.97   628.2  824.81   637.8  828.27   647.5  832.29   686.3  850.05
     696  853.76   705.7  856.46   725.1  860.21   734.8  861.59   812.4  868.86
#Mann= 3 , 0 , 0
       0     .06       0   390.6    .045       0   405.6      .1       0
Bank Sta=390.6,405.6
XS Rating Curve= 0 ,0
Exp/Cntr=0.3,0.1

Type RM Length L Ch R = 1 ,52290.1 ,515.1,515.9,514.3
XS GIS Cut Line= 3
      1831053.42      655262.582     1831482.424      655113.021
     1831840.583      655057.919
#Sta/Elev= 30
       0  816.54     9.7  813.92    77.3  799.18   164.3  778.43   183.7  775.02
     232  770.89   251.3   769.7   338.3  767.73   386.7  765.54   431.4  762.87
     435  762.67   444.7  763.02   446.4  763.52   454.3  765.83   483.7  782.69
   503.3  793.21   513.1  797.88   552.3  814.27   581.6  827.95   601.2  838.03
     611  843.66   630.6   856.3   640.4  861.62   650.2  865.37     660  867.99
   689.4  874.41   728.6  885.53   748.1  889.79   767.7  892.83   816.7  898.46
#Mann= 3 , 0 , 0
       0     .06       0   431.4    .045       0   446.4      .1       0
Bank Sta=431.4,446.4
XS Rating Curve= 0 ,0
Exp/Cntr=0.3,0.1

Type RM Length L Ch R = 1 ,51774.1 ,597.3,585.3,572
XS GIS Cut Line= 3
     1831025.467      655679.943     1831322.689      655691.054
     1831842.134       655496.61
#Sta/Elev= 30
       0  888.71    38.4  873.18    86.4  852.58      96  847.42   105.5  840.61
   115.1  833.01   124.7  826.42   134.3  821.42   163.1  810.25   191.9  801.59
     259  787.76   307.2  775.84   336.4  771.18   394.7  766.19   501.8  761.86
   531.2  759.68   540.7   759.5   546.2  759.62   608.8  762.45   618.5  764.18
   628.3  768.06     638  773.51   667.2   791.6   676.9  796.96   715.8  813.54
   754.8  832.37     784  845.35   813.2  860.24   822.9   864.1   852.1  873.75
#Mann= 3 , 0 , 0
       0     .07       0   531.2    .045       0   546.2     .08       0
Bank Sta=531.2,546.2
XS Rating Curve= 0 ,0
Exp/Cntr=0.3,0.1

Type RM Length L Ch R = 1 ,51188.9 ,527.8,525.3,522.4
XS GIS Cut Line= 3
     1831657.454      656375.245     1831945.053       656014.04
     1832145.496      655745.514
#Sta/Elev= 30
       0  848.84    19.6  835.91    39.3  822.13    49.1  815.91    58.9  810.79
    68.8   806.6    88.4  799.96   127.7  788.94   186.6  774.82     226  764.33
   235.8  762.84   245.6  762.32   324.2  761.19     393  759.07   454.2  757.98
   461.7  757.94   469.2  758.66   471.3  758.86   480.9  761.44     500  769.22
   528.7  779.75   586.2  797.22   595.8  800.41   614.9  807.98   624.5  812.45
     634  817.57   681.9  846.34   710.6  862.29   739.4  876.67   796.8  902.26
#Mann= 3 , 0 , 0
       0     .06       0   454.2    .045       0   469.2      .1       0
Bank Sta=454.2,469.2
XS Rating Curve= 0 ,0
Exp/Cntr=0.3,0.1

Type RM Length L Ch R = 1 ,50663.6 ,238.9,253,256.7
XS GIS Cut Line= 3
     1832157.605      656641.287     1832393.153      656244.532
     1832496.086      655972.198
#Sta/Elev= 30
       0  859.51    19.6  856.92    29.4  854.88    39.3  851.63    49.1  847.27
    68.7  837.58    98.2  821.91   137.4  800.29   166.9  785.16   186.5   776.3
   196.3   772.4   206.2  768.74   225.8   762.6   245.4  758.41   265.1  755.98
   274.9   755.4   369.4  754.88   384.4  754.95     432  755.36   441.8   756.3
   451.6  758.35   461.4  761.19   548.8  788.18   568.2  796.25   597.3  810.08
   616.7  819.87   665.2  845.68     704  865.81   733.1  880.16   752.6  888.94
#Mann= 3 , 0 , 0
       0     .06       0   369.4    .045       0   384.4     .08       0
Bank Sta=369.4,384.4
XS Rating Curve= 0 ,0
Exp/Cntr=0.3,0.1

Type RM Length L Ch R = 1 ,50410.6 ,120,109.9,108.6
XS GIS Cut Line= 2
     1832276.533      656745.334     1832830.451      656080.972
#Sta/Elev= 30
       0  843.33    19.7  844.57    39.3  844.58      59  843.08    68.8  841.49
    78.6  838.92    88.5   835.4    98.3   831.1   186.8   790.9   245.7   767.9
   265.4   760.7   275.2  757.74     285  755.81   294.9  754.93   383.4  754.24
   419.8  752.72   422.7  752.65   434.8  752.76   501.3  754.58   530.8  754.54
   550.4  755.64   570.1  758.36   589.8  762.12   619.2  768.84   658.6  775.38
   678.2  778.11   707.7  781.08     747  786.81     806   792.8     865  794.44
#Mann= 3 , 0 , 0
       0     .06       0   419.8    .045       0   434.8     .07       0
Bank Sta=419.8,434.8
XS Rating Curve= 0 ,0
Exp/Cntr=0.3,0.1

Type RM Length L Ch R = 1 ,50300.8 ,385,404.9,421.9
XS GIS Cut Line= 2
     1832355.772      656818.839      1832909.69      656154.477
#Sta/Elev= 30
       0  819.86    29.5  810.68    39.3  808.24    49.2  806.82    68.8   804.9
   127.8  800.35   167.1  794.06   186.8  790.11   196.6  787.62   206.4  784.57
   216.2  780.83   265.4  759.94   275.2  756.89     285  755.03   294.9  754.19
   314.5  753.61   373.5  754.22     403  753.95   422.7  752.98     437  751.52
   442.3  751.16     452  751.38   471.8  753.09   481.6  753.38     521  753.93
   609.4  756.56   697.9  758.35   776.5  762.26   845.3  764.96     865  765.45
#Mann= 3 , 0 , 0
       0     .06       0     437    .045       0     452     .06       0
Bank Sta=437,452
XS Rating Curve= 0 ,0
Exp/Cntr=0.3,0.1

Type RM Length L Ch R = 1 ,49895.9 ,697,706.9,702.6
XS GIS Cut Line= 3
     1832389.755      656847.724      1832595.35      656727.086
     1833281.627      656709.927
#Sta/Elev= 30
       0  814.43    38.1  801.09    57.2  795.28    66.8  792.76    76.3  790.76
   104.9  786.07   114.4     784     124  781.62   162.1  770.06   181.2  765.93
   200.2  763.03   248.2  757.59   297.2  756.29   478.1  749.77   483.6  749.65
   493.1  749.68   522.8  750.21   591.4  752.48   620.8  752.61   650.3  752.22
   660.1  752.98   669.9  754.85   679.7  757.35   758.2  779.44     817  795.31
   846.4  802.72     866  806.47   875.8  808.84   895.4  815.64   924.9  824.02
#Mann= 3 , 0 , 0
       0     .06       0   478.1    .045       0   493.1     .07       0
Bank Sta=478.1,493.1
XS Rating Curve= 0 ,0
Exp/Cntr=0.3,0.1

Type RM Length L Ch R = 1 ,49189   ,937.8,931.6,932
XS GIS Cut Line= 3
     1832469.162      657320.032      1833014.96      657284.927
     1833370.464      657323.968
#Sta/Elev= 30
       0  791.25    19.5  786.74    48.8  780.65   107.4  769.75   156.3  761.92
     166   760.6   185.6  758.41   195.3   757.6   214.9  756.48   273.5  753.84
   400.4  749.82   439.5  748.31   478.4  747.22   488.3  747.12   493.4  747.38
   498.1  747.62   507.9  749.33   537.2   757.7   624.2  783.39   691.9  804.52
   701.6  807.75   711.2  811.73   720.9  816.51   730.6  821.68   759.6  837.61
   817.6  870.48   836.9  880.94   856.2  890.47   865.9  894.84   904.6  911.02
#Mann= 3 , 0 , 0
       0     .06       0   478.4    .045       0   493.4      .1       0
Bank Sta=478.4,493.4
XS Rating Curve= 0 ,0
Exp/Cntr=0.3,0.1

Type RM Length L Ch R = 1 ,48257.4 ,479.6,469.7,456.3
XS GIS Cut Line= 3
     1832427.238      658043.942     1832898.129      658056.696
      1833328.54      658000.648
#Sta/Elev= 30
       0  824.69    39.3  808.48    68.7  797.05    98.1  786.82   117.8  781.32
   176.6  769.55   206.1  762.98   225.7  757.95   235.5  755.77   245.4  754.06
   255.2  752.84   362.7  742.01   372.9  741.83   377.7  741.91   412.2  742.46
   461.2  742.65   490.4  743.38     500  743.99   548.2   748.4   567.5  750.67
   586.8   753.9   606.1  758.16     635  765.86   702.6  785.79   770.1  804.53
   779.7  808.22   789.4   812.9     828  833.18   885.8  864.75   905.1  875.03
#Mann= 3 , 0 , 0
       0     .06       0   362.7    .045       0   377.7     .08       0
Bank Sta=362.7,377.7
XS Rating Curve= 0 ,0
Exp/Cntr=0.3,0.1

Type RM Length L Ch R = 1 ,47787.7 ,609.1,602.9,596
XS GIS Cut Line= 3
      1832052.46      659066.177      1832596.21      658666.177
      1833464.96      658151.593
#Sta/Elev= 30
       0  904.06   117.4  883.61   185.9  873.72     225  870.34   254.4  866.03
   283.7  858.83   342.4  846.87   371.8  838.85   401.1   829.9   498.9  796.64
   518.5  790.99   635.9  765.88   684.8   757.7   714.2  755.36   792.7  752.56
   900.5  752.74  1018.1  744.85  1096.6  741.06  1248.3  740.56  1253.4  740.53
  1263.3  741.09    1273  743.14  1351.4  764.56  1478.9  796.92  1488.7  800.14
  1508.3  809.31  1606.3   860.8  1616.1  865.33  1645.5   876.4  1684.7  895.57
#Mann= 3 , 0 , 0
       0     .06       0  1248.3    .045       0  1263.3     .08       0
Bank Sta=1248.3,1263.3
XS Rating Curve= 0 ,0
Exp/Cntr=0.3,0.1

Type RM Length L Ch R = 1 ,47184.8 ,442.8,441.6,439.5
XS GIS Cut Line= 3
     1833095.672      659155.346     1833397.638      658842.299
     1833670.301      658596.459
#Sta/Elev= 30
       0  785.86      29  778.74    96.7  762.72   106.3  760.73     116  759.15
   164.3  753.57   212.6   748.5   241.6  745.56   280.3  742.14   299.6  740.77
     319  739.72   338.3     739   368.9  738.38     377  738.24   383.9  738.64
   386.6   738.8   396.3  740.45   415.6  744.98   483.3   758.2   512.2  764.26
   531.6  768.62   541.2  770.34   579.9  775.46   628.2  782.85   686.1  792.89
   705.5  796.46   715.1  798.48   724.8  801.22   734.4  805.22   802.1  837.72
#Mann= 3 , 0 , 0
       0     .06       0   368.9    .045       0   383.9     .08       0
Bank Sta=368.9,383.9
XS Rating Curve= 0 ,0
Exp/Cntr=0.3,0.1

Type RM Length L Ch R = 1 ,46743.2 ,1037,1042.8,1046
XS GIS Cut Line= 3
     1833267.043       659537.01     1833694.127      659116.177
      1834002.46      658834.927
#Sta/Elev= 30
       0  839.54    29.5     832    49.2  825.65    98.3  803.99   127.8  792.65
   157.3  782.88   186.8  775.24   235.9  766.37     285  759.01   314.5  756.67
   393.2  752.76     462  739.66   479.1  737.39   491.5  736.93   494.1  737.06
     521  739.23   540.6   742.7   560.3  748.25   589.8  758.12   609.3  763.87
   628.7  768.06   648.1  771.48   667.5  774.61   696.6  778.49   803.4  789.19
   842.2   794.7   851.9  796.62   861.6  799.55   890.8  811.32  1016.9  864.71
#Mann= 3 , 0 , 0
       0     .06       0   479.1    .045       0   494.1     .07       0
Bank Sta=479.1,494.1
XS Rating Curve= 0 ,0
Exp/Cntr=0.3,0.1

Type RM Length L Ch R = 1 ,45700.4 ,687.5,683,678.6
XS GIS Cut Line= 4
      1833908.71      660053.677     1834087.336        659746.8
      1834458.71      659426.593      1834571.21      659178.677
#Sta/Elev= 30
       0  869.01    38.4  855.32      48  852.48   105.6  837.74   115.2  834.64
   124.8  830.73   172.7  808.41   191.9  800.29   211.1  793.08   230.3  787.22
   268.7  777.17   287.9   772.9   326.3  765.48   413.9  749.78   433.5  747.04
   580.6   737.7   695.1  731.72   698.3  731.69   710.1  732.66   757.2  741.35
     816  753.86   855.2  760.94  1010.7  794.34  1020.4   797.7  1030.2  802.51
  1049.6  814.47  1059.4  819.99  1069.1  824.78  1088.5  832.42  1117.7  841.99
#Mann= 3 , 0 , 0
       0     .06       0   695.1    .045       0   710.1     .08       0
Bank Sta=695.1,710.1
XS Rating Curve= 0 ,0
Exp/Cntr=0.3,0.1

Type RM Length L Ch R = 1 ,45017.4 ,756.7,765.5,773.4
XS GIS Cut Line= 4
     1834537.877      660572.427      1834577.46      660197.427
     1834850.377      659857.843     1835356.627       659743.26
#Sta/Elev= 30
       0  849.68    19.3  846.74    67.7  837.24    96.7  829.48   106.4  825.42
     116  817.44   125.7  806.12   135.4  796.31     145  791.47     174  786.46
   261.1  762.68   328.7  743.38   348.1  740.79   454.5  736.62   522.3  733.24
   546.2  731.37   551.4  731.17   561.2   732.2   580.4  735.95   590.1  736.92
   725.6  741.54   842.1  743.45   910.7  746.72   959.6  751.47  1028.2  762.57
  1096.8  778.49  1135.9  790.28  1194.7  813.34  1292.6  854.72  1331.8  869.26
#Mann= 3 , 0 , 0
       0     .06       0   546.2    .045       0   561.2     .06       0
Bank Sta=546.2,561.2
XS Rating Curve= 0 ,0
Exp/Cntr=0.3,0.1

Type RM Length L Ch R = 1 ,44251.9 ,448.4,447.4,447.2
XS GIS Cut Line= 2
     1834773.293      660797.427     1835494.127      660376.593
#Sta/Elev= 30
       0  834.17    29.5  830.89    39.3  828.85    49.1  825.31    58.9   820.7
    68.7  815.54    98.2  798.45     108  793.21   117.8   788.6   157.1  773.01
   206.2  751.12   225.9  743.45   245.5  736.97   255.3  735.19   265.1  734.74
   402.6  732.83   412.4  732.44     427  730.61   432.1  729.95   441.9  729.76
     442  729.78   451.7  731.26   471.4   735.7     599  755.83   667.8  767.24
   746.3  780.98     766  785.91   805.2  797.16   824.9  803.81   834.7  808.14
#Mann= 3 , 0 , 0
       0     .06       0     427    .045       0     442     .06       0
Bank Sta=427,442
XS Rating Curve= 0 ,0
Exp/Cntr=0.3,0.1

Type RM Length L Ch R = 1 ,43804.4 ,833.2,852.8,871.2
XS GIS Cut Line= 3
     1834979.284      661192.685     1835263.229       661006.53
      1835632.63      660775.489
#Sta/Elev= 30
       0  832.22    19.4   829.3    67.9  826.03    87.3  823.73      97  820.67
   106.7  813.55   116.4  803.43   126.1  792.07   135.8  782.43   145.5  777.59
   184.3  765.95     194  762.07   213.4  751.18   223.1  746.98   232.8  745.14
   242.5  744.17   281.3  735.01     291  733.53     332  729.35   339.5  729.06
     347  729.62   368.6  732.39   387.9   733.7   552.5  740.46   581.6     742
   591.3  742.97   620.3  748.11   755.9  774.09   765.6  776.13   775.2  779.16
#Mann= 3 , 0 , 0
       0     .06       0     332    .045       0     347     .06       0
Bank Sta=332,347
XS Rating Curve= 0 ,0
Exp/Cntr=0.3,0.1

Type RM Length L Ch R = 1 ,42951.6 ,858.5,853,845.6
XS GIS Cut Line= 3
      1834864.96      661745.691     1835248.641      661651.941
     1835932.668      661822.079
#Sta/Elev= 30
       0  848.31    19.3  843.93    38.5  838.54    77.1  824.77     106  815.61
   115.6  811.59   163.8  787.45   173.4  783.15   221.6  764.39   240.8  758.54
   250.5  757.08   279.4  754.28   317.9   748.5   375.7  742.46   434.1  733.64
   502.7  728.76   520.8  725.56     532  724.19   535.8  724.28     581  727.84
   688.7  730.23     767  732.84   864.9  738.12   884.5  739.94   923.6  749.29
     953  757.28  1011.7  778.99  1041.1  790.32  1060.7  799.02  1099.8   821.6
#Mann= 3 , 0 , 0
       0     .08       0   520.8    .045       0   535.8     .06       0
Bank Sta=520.8,535.8
XS Rating Curve= 0 ,0
Exp/Cntr=0.3,0.1

Type RM Length L Ch R = 1 ,42098.7 ,408.1,409,409.2
XS GIS Cut Line= 3
     1834913.571      662221.385     1835094.127      662327.288
      1835825.03      662226.593
#Sta/Elev= 30
       0  801.56     9.5  801.16      19   799.8    28.5  796.83    57.1     784
    76.1  776.65   142.7  753.56   152.2  751.02   180.8  747.69   190.3  746.19
   248.7  735.37   258.5  734.08     288  732.17   415.9  726.53   445.4  724.38
   455.2  723.92   465.1  724.38   474.9   725.6   494.6  726.81   583.1  727.94
   671.7  729.78   691.4  731.48   730.7  738.84   740.5  741.22   789.7  760.53
   848.8  785.84   897.9   808.9   907.8  813.12   927.4  820.59   947.1  827.42
#Mann= 3 , 0 , 0
       0     .06       0   445.4    .045       0   474.9     .06       0
Bank Sta=445.4,474.9
XS Rating Curve= 0 ,0
Exp/Cntr=0.3,0.1

Type RM Length L Ch R = 1 ,41689.6 ,893.5,894.8,883.3
XS GIS Cut Line= 4
     1834772.946      662879.371     1835094.127      662704.024
     1835821.557      662620.691     1836054.196      662636.316
#Sta/Elev= 30
       0  845.44    28.9  844.47      77   837.4   105.9  829.97   125.2  821.46
   134.8   818.9     183  809.48   240.7  794.76     260  788.36   269.6  783.29
   298.5  760.64   308.2  755.44     337  744.48   356.3  740.08   512.4  728.22
   570.9  725.05   775.4  722.22     776   722.2   790.4  723.16     815  726.49
   951.7  736.93  1010.2  748.82  1078.6  768.15  1098.1  775.34  1107.8  780.63
  1166.1  818.56  1195.3  832.28    1273  850.83  1302.1  854.71  1331.3   856.3
#Mann= 3 , 0 , 0
       0     .06       0   775.4    .045       0   790.4     .07       0
Bank Sta=775.4,790.4
XS Rating Curve= 0 ,0
Exp/Cntr=0.3,0.1

Type RM Length L Ch R = 1 ,40794.8 ,750.7,752.5,754.2
XS GIS Cut Line= 2
     1835176.075      663278.669     1835868.779      663207.824
#Sta/Elev= 30
       0  838.56     9.8  837.82    19.6  836.37    29.4  833.36    39.2  828.57
    88.3  799.41   107.9  788.48   176.5  754.71   186.3  750.99   196.2  749.15
     206     748   215.8  745.89     255  732.54   274.6  724.44   284.4   721.1
   291.1  720.49   294.2  720.21   306.1  721.66   313.8  722.79   323.6  723.21
   372.7   722.9   421.7  723.24     510  725.54   519.8  726.75   529.6  729.93
   539.4  734.29   637.5   780.2   647.3  785.28   657.1  791.05   696.3  815.91
#Mann= 3 , 0 , 0
       0     .08       0   291.1    .045       0   306.1     .06       0
Bank Sta=291.1,306.1
XS Rating Curve= 0 ,0
Exp/Cntr=0.3,0.1

Type RM Length L Ch R = 1 ,40042.3 ,574.5,567.3,560.2
XS GIS Cut Line= 2
     1835164.268      663891.738     1835904.201      663883.867
#Sta/Elev= 30
       0  836.55    19.5  825.85    87.6  785.47   155.8  746.88   165.5  743.63
   175.3  742.41     185  740.24   194.7  736.95   204.5  734.88   253.2  729.16
   301.8  724.25   327.4  719.45     331  718.96   342.4  719.35   399.2  725.31
   428.4  727.11   438.1  729.13   477.1   741.3   496.6  745.47   525.8   749.4
   564.7   752.8   584.2  756.51   603.7  762.98   632.9  774.02   642.6  779.18
   652.4  786.67   662.1  795.64   671.8  803.34   681.6  808.07     740  821.93
#Mann= 3 , 0 , 0
       0     .06       0   327.4    .045       0   342.4     .06       0
Bank Sta=327.4,342.4
XS Rating Curve= 0 ,0
Exp/Cntr=0.3,0.1

Type RM Length L Ch R = 1 ,39475   ,477.8,479.4,480.2
XS GIS Cut Line= 3
     1834976.071       664587.01     1835740.655      664309.927
     1835894.821       664280.76
#Sta/Elev= 30
       0  837.59    19.6   837.7    39.2  836.41      49  834.98    58.8  832.02
   156.8  777.82   176.4  768.37     245  738.82   313.5  729.93   333.1  728.28
   382.1  726.69   450.7  727.36   499.7  726.63   548.7  724.63   558.5  723.49
     572  720.13     587  717.57   587.9  717.47   617.3  719.56   754.4  723.19
   764.2  724.21     774  726.88   813.2  745.19   832.8  755.46   842.7  762.47
   872.1  790.19   881.9  798.24   891.7  803.79   950.5  824.99   970.1  826.74
#Mann= 3 , 0 , 0
       0     .07       0     572    .045       0     587     .06       0
Bank Sta=572,587
XS Rating Curve= 0 ,0
Exp/Cntr=0.3,0.1

Type RM Length L Ch R = 1 ,38995.6 ,575.8,927.6,927.2
XS GIS Cut Line= 4
     1835014.707       665065.53     1835228.155      664891.177
     1835982.321      664676.593     1836203.155       664574.51
#Sta/Elev= 30
       0  840.72      57  827.63   142.6  801.02   152.1  796.97   161.6  791.87
   209.1  764.23   228.1  754.03   247.1  745.13   256.6  741.33   266.1  738.62
   285.4  737.35   314.8  732.45   344.2  729.79   373.6  728.86     403  729.68
   481.4  727.02   540.2  726.24   579.4  723.08   633.6  716.79     648  716.48
   648.6  716.49   775.5  720.75   863.7  729.45   971.5   734.9  1020.5  735.32
  1040.1  737.76  1147.3  764.63  1166.8  770.77  1225.1   801.9    1303  835.74
#Mann= 3 , 0 , 0
       0     .06       0   633.6    .045       0   648.6     .06       0
Bank Sta=633.6,648.6
XS Rating Curve= 0 ,0
Exp/Cntr=0.3,0.1

Type RM Length L Ch R = 1 ,38068   ,1316.3,980.8,990.6
XS GIS Cut Line= 3
     1835051.071      665195.343     1835367.738       665293.26
     1836330.238       664912.01
#Sta/Elev= 30
       0  816.62    29.2  804.52      39  799.51    48.7  792.85      78  768.76
    87.7  761.55    97.5  755.39   107.2  751.24   126.7  748.59   136.5  746.44
   165.7  737.06   185.2  732.28   214.5  727.71   243.7   726.4   321.7  727.24
   438.9  726.08   526.8  723.27   702.6  721.45   897.9  717.12  1015.1  717.32
    1069  716.62  1073.7  716.52    1084  716.74  1093.2  718.36  1122.6  727.08
  1161.6   737.1  1200.7  740.24    1230  745.03  1298.4  759.83  1366.7  777.84
#Mann= 3 , 0 , 0
       0     .06       0    1069    .045       0    1084     .08       0
Bank Sta=1069,1084
XS Rating Curve= 0 ,0
Exp/Cntr=0.3,0.1

Type RM Length L Ch R = 1 ,37087.1 ,147.1,147.2,147.1
XS GIS Cut Line= 3
     1835067.738       665705.76     1835613.571       665518.26
     1836815.655       665530.76
#Sta/Elev= 30
       0  722.26    68.5  719.74   156.5  720.77   185.9  725.29   205.4  726.16
   283.7  724.16   352.2  719.91   401.1  720.15     450  724.04   489.1  720.03
   518.4  718.89   577.1  719.49   606.5  723.29   655.3  725.18   674.9  723.89
   704.2  718.58   899.7   718.1   958.3  713.04   997.4  715.42  1026.5  714.97
  1041.5  714.41  1075.6  717.99  1202.6  720.01  1437.2  718.18  1515.4  724.16
  1622.9  724.87  1642.5     727  1671.8  735.66  1691.3  738.88  1779.3     745
#Mann= 3 , 0 , 0
       0     .06       0  1026.5    .045       0  1041.5     .06       0
Bank Sta=1026.5,1041.5
XS Rating Curve= 0 ,0
Exp/Cntr=0.3,0.1

Type RM Length L Ch R = 1 ,36940   ,719.1,715.3,710.3
XS GIS Cut Line= 3
     1835094.821      665851.593     1835640.655      665664.093
     1836842.738      665676.593
#Sta/Elev= 30
       0  729.57    48.9  727.06   117.4  727.15   234.8  729.95   273.9  736.91
   303.2  745.77   342.4  755.34   361.9  758.53   391.3  759.82   430.4  754.68
   498.9   749.9   508.7   748.4     538   740.8   547.8  739.52   665.1  735.82
   753.1  727.64   831.2  725.11   860.6   719.4   919.2  717.88     983  713.68
   997.4  712.97     998     713  1046.3  718.05  1095.1     720  1202.6  718.74
  1593.6  718.54  1622.9  725.38  1632.7  726.35  1740.2  728.82  1779.3  727.09
#Mann= 3 , 0 , 0
       0     .06       0     983    .045       0     998     .06       0
Bank Sta=983,998
XS Rating Curve= 0 ,0
Exp/Cntr=0.3,0.1

Type RM Length L Ch R = 1 ,36224.7 ,330.6,329.9,329.2
XS GIS Cut Line= 5
     1835657.321       665993.26     1836176.071      665989.093
     1836630.238      665895.343     1836832.321      665782.843
     1837003.155      665701.593
#Sta/Elev= 30
       0  793.85    29.4  785.56    97.9   764.3   117.5  759.07   215.3  740.31
   244.7  733.97   264.3  731.32   332.8  726.85   391.5  723.94   430.7  722.33
   469.8  722.12     509  720.88   576.7  717.15     683  715.83   779.6   715.6
   856.9  714.58   871.3  713.77   885.9  713.15   886.3   713.2   924.5  718.48
   953.5  721.06   992.2  723.26  1011.4  723.05  1040.3  720.93  1059.6  720.53
  1098.2  721.74    1156  725.85  1194.5  727.28  1346.2   724.4    1403  724.38
#Mann= 3 , 0 , 0
       0     .06       0   871.3    .045       0   886.3     .06       0
Bank Sta=871.3,886.3
XS Rating Curve= 0 ,0
Exp/Cntr=0.3,0.1

Type RM Length L Ch R = 1 ,35894.8 ,1309.2,1313,1292.5
XS GIS Cut Line= 4
     1836031.433      666393.996     1836217.738      666322.427
     1836778.155      666191.177     1837111.488       666162.01
#Sta/Elev= 30
       0  788.88     9.5  783.31      38  766.09    47.5   760.7      57  756.41
    66.5   753.4     114  741.41   152.1  732.06   199.6  720.11   209.3  717.79
   219.1  716.04   228.8  715.35   258.1  715.06   453.2  714.78     541  714.33
   550.8  714.19   570.3   712.9   574.1  712.83     580  712.71   589.1  712.78
   609.3   713.7   638.6  714.19   677.6  715.49   706.9  716.63   765.4   719.2
   794.8  722.05   912.9  729.56     972  732.95   991.7  734.28  1109.8  746.52
#Mann= 3 , 0 , 0
       0     .06       0   574.1    .045       0   589.1     .06       0
Bank Sta=574.1,589.1
XS Rating Curve= 0 ,0
Exp/Cntr=0.3,0.1

Type RM Length L Ch R = 1 ,34581.7 ,1182.8,1177,1168.5
XS GIS Cut Line= 2
     1836157.475      667055.455     1837068.933      667263.788
#Sta/Elev= 30
       0  787.58    19.7  778.25    78.7  751.79    88.6  748.74   157.5  734.04
   275.6  714.03   295.2  712.77   334.6  712.53     374  712.71   423.2     714
     433  713.88   472.4  711.18   492.1  712.35   501.9  712.34   519.3  711.05
   531.4  710.81   551.1  711.27   629.9  718.56   669.2  722.88   708.6  729.81
   757.8  736.17   777.5  740.87     807  749.71   836.6  757.81   856.2  761.27
   875.9  763.44   895.6  766.29   915.3  768.11   925.1  771.25     935  775.93
#Mann= 3 , 0 , 0
       0     .06       0   519.3    .045       0   551.1     .06       0
Bank Sta=519.3,551.1
XS Rating Curve= 0 ,0
Exp/Cntr=0.3,0.1

Type RM Length L Ch R = 1 ,33404.7 ,787.8,783,778
XS GIS Cut Line= 2
       1836110.6       668158.58     1836943.933      667866.913
#Sta/Elev= 30
       0  796.57    39.2  775.29    58.9  765.23    78.5  755.99    98.1  747.91
   117.7  740.94   137.3  734.84     206  716.89   225.6  710.44   235.4  708.84
   245.2  708.95   251.8  709.68   264.9  711.06   274.7  711.17   304.1   710.3
   353.2  710.48   451.3  713.62   549.4  713.48   559.2  713.73     569  714.97
   608.2  724.83   716.1  745.06   745.6  753.08   755.4   754.5   784.8  754.83
   794.6  756.18   804.4  759.12   814.2  762.88   863.3   785.1   882.9  795.08
#Mann= 3 , 0 , 0
       0     .08       0   225.6    .045       0   251.8     .06       0
Bank Sta=225.6,251.8
XS Rating Curve= 0 ,0
Exp/Cntr=0.3,0.1

Type RM Length L Ch R = 1 ,32621.7 ,625.4,606,584.6
XS GIS Cut Line= 3
     1836190.655      668726.593     1836498.988       668662.01
     1837057.321      668328.677
#Sta/Elev= 30
       0  820.47    38.2  814.95    47.7  812.07    66.8  803.59    95.5  794.94
     105  789.36   124.1  774.49   133.6  769.08   162.3  757.31   171.8  752.94
   190.9  742.62   200.5  739.22     315  719.46   334.4  716.89   392.7  712.83
     645  708.48   674.1  708.42   693.5  709.36   712.9  708.35   722.6  707.51
   732.4  707.53   742.1  709.34   771.2  721.19   790.6  727.68   800.3  729.21
   829.4  731.87   848.8  736.69   887.6  748.13   926.5   756.3   965.3  765.46
#Mann= 3 , 0 , 0
       0     .06       0   712.9    .045       0   742.1     .08       0
Bank Sta=712.9,742.1
XS Rating Curve= 0 ,0
Exp/Cntr=0.3,0.1

Type RM Length L Ch R = 1 ,32015.6 ,467.7,400.7,376.9
XS GIS Cut Line= 2
     1836990.808      669347.121     1837355.392      668420.038
#Sta/Elev= 30
       0  763.76     9.8  760.35    19.5  758.02    87.9     743   117.2  740.31
     166  732.29   185.6  727.77   214.9  719.53   234.4  715.38   244.2  714.24
   253.9  713.86   302.8  712.92   380.9  709.81   406.6  707.33     420  707.01
   429.7  707.51     459  709.54   576.2   709.4   615.3   710.6   664.1  712.94
   673.9  714.57   693.4  719.73   722.7  722.86   742.3  728.03   771.6  731.11
   859.5  741.71     879  744.98   918.1  753.31   937.6  756.73   996.2  763.79
#Mann= 3 , 0 , 0
       0     .06       0   406.6    .045       0   429.7     .06       0
Bank Sta=406.6,429.7
XS Rating Curve= 0 ,0
Exp/Cntr=0.3,0.1

Type RM Length L Ch R = 1 ,31614.9 ,172.6,218.4,222.2
XS GIS Cut Line= 5
     1837497.599      669457.843     1837494.127      669264.788
     1837379.543       669055.76     1837351.766      668935.968
     1837351.766      668590.135
#Sta/Elev= 30
       0  782.76    77.2  750.69    96.5  743.25   115.8  736.47   173.8  717.64
   183.4  715.37   193.1  714.04   202.6  713.47   212.2  712.35   231.2  708.21
   240.8  706.64   250.3  705.64   278.9  704.72   307.5  705.08   326.6  706.28
   345.6  708.16   355.2  708.71   421.9  710.87   459.8  711.48   535.5  710.26
   573.6  710.44   602.5   711.3   650.5  713.78   708.1  714.57   746.6  715.88
   765.8  717.41   775.4  719.09   804.2  725.41   813.8  726.96   900.3  736.88
#Mann= 3 , 0 , 0
       0     .08       0   278.9    .045       0   326.6     .06       0
Bank Sta=278.9,326.6
XS Rating Curve= 0 ,0
Exp/Cntr=0.3,0.1

Type RM Length L Ch R = 1 ,31396.5 ,259.4,291.9,323.6
XS GIS Cut Line= 6
     1837667.043      669481.802     1837668.432      669294.302
     1837530.932      669122.079     1837486.488      668988.746
     1837462.877      668887.357     1837461.488      668617.913
#Sta/Elev= 30
       0  757.06    46.9  745.02      75  737.24     150  714.53   159.4   712.9
   168.8   712.3   216.2  711.34   225.8  710.77   235.4  709.68   247.4  707.25
   254.6  705.95   264.2  704.98   273.7  705.18   283.3  706.95   292.9  709.21
   302.5  710.22   398.3  710.36     436   711.2   529.7   712.1   586.3  713.64
   624.1  714.08   719.9  713.31     768     714   777.6  714.81   787.3  716.93
   816.1  726.19     845   737.3   854.6   739.2   873.9  740.07     922  740.43
#Mann= 3 , 0 , 0
       0     .06       0   247.4    .045       0   283.3     .06       0
Bank Sta=247.4,283.3
XS Rating Curve= 0 ,0
Exp/Cntr=0.3,0.1

Type RM Length L Ch R = 1 ,31104.6 ,502.7,509.5,516.2
XS GIS Cut Line= 3
     1837693.432      669485.621     1838061.488       669062.01
     1838466.002      668865.829
#Sta/Elev= 30
       0  751.87    87.1  721.98   106.4  716.19   116.1  713.89   125.8  712.85
   145.1  712.33   193.5  709.65   215.9  705.87   222.5   704.9   232.2  704.34
   241.9  704.49   251.6  705.23   270.9  707.19   309.6  707.59     329  708.13
   377.3  710.92   493.4  714.27   570.9  715.83   619.8   717.3   707.8   720.9
   766.4  724.27     786  726.74   805.5  729.62   873.9  741.26   883.7  743.44
   942.3  757.97   981.4  766.65   991.2  769.37    1001   773.2  1010.8  777.63
#Mann= 3 , 0 , 0
       0     .06       0   215.9    .045       0   251.6     .06       0
Bank Sta=215.9,251.6
XS Rating Curve= 0 ,0
Exp/Cntr=0.3,0.1

Type RM Length L Ch R = 1 ,30595.1 ,486.3,489.8,492.6
XS GIS Cut Line= 2
     1837865.808      669737.746     1838626.225       669102.33
#Sta/Elev= 30
       0  779.48    49.1  756.46    58.9  752.11    68.7  748.82    98.1  746.05
   107.9  744.08     157  730.61     206  718.69   215.8  716.77   235.5  714.28
   255.1  713.36   274.7  711.15   284.5  710.65   372.8  708.87   441.5   706.4
   452.8  705.01   461.1  704.25     471  704.44   480.8  705.85   490.6  707.48
   500.4  708.04   627.9   710.9   647.6  713.63   696.6  724.37   745.7  731.59
   824.2  747.91   902.6  764.72   912.5  767.27   922.3  771.08     991  800.95
#Mann= 3 , 0 , 0
       0     .06       0   452.8    .045       0   480.8     .06       0
Bank Sta=452.8,480.8
XS Rating Curve= 0 ,0
Exp/Cntr=0.3,0.1

Type RM Length L Ch R = 1 ,30105.4 ,453.2,462.9,472.5
XS GIS Cut Line= 3
     1838055.901      669897.698     1838642.012      669553.254
     1838786.457      669414.365
#Sta/Elev= 30
       0  756.59    19.4  752.34    38.8  745.86    87.4  728.21   116.5  719.64
   126.2  717.68   145.7  715.78   165.1  711.54   174.8  710.38   330.2  708.41
   456.5  709.66   524.4  709.24   534.2  709.03   543.9  707.94   553.6  705.77
   563.3  704.31     573  704.37   582.7   705.5   592.4  707.03   611.8  708.95
   621.6  710.46   650.7  716.22   660.4  717.65   679.8  719.26   689.4  721.57
   746.6  743.83   784.8  756.66   803.9  763.75   851.6  783.89   880.2  798.38
#Mann= 3 , 0 , 0
       0     .06       0   553.6    .045       0   582.7     .06       0
Bank Sta=553.6,582.7
XS Rating Curve= 0 ,0
Exp/Cntr=0.3,0.1

Type RM Length L Ch R = 1 ,29642.5 ,116.8,115.4,112.6
XS GIS Cut Line= 3
     1838102.022      669985.621     1838439.053      669946.908
     1838761.282      669682.749
#Sta/Elev= 30
       0  746.69    19.4  742.11    58.2  734.56    77.5   730.5    87.2  728.03
   106.6  722.52   116.3  720.19   135.7  717.02   155.1  710.71   164.8  709.51
   242.3  709.21     252   708.3   261.7  706.13   271.4  704.11   281.1  703.95
   290.8  705.59   300.5  707.53   310.2  708.58   339.2  709.86     378  710.05
   445.8  712.82   494.3  713.34   523.4  714.33   552.4  715.99   571.8  717.58
   610.6  721.53   649.3  724.11   668.7  725.85   707.5   730.8   755.9  737.67
#Mann= 3 , 0 , 0
       0     .06       0   261.7    .045       0   290.8     .06       0
Bank Sta=261.7,290.8
XS Rating Curve= 0 ,0
Exp/Cntr=0.3,0.1

Type RM Length L Ch R = 1 ,29527.1 ,676.6,667.8,660
XS GIS Cut Line= 3
     1838152.947      670110.318     1838485.309      670033.323
     1838810.242      669744.234
#Sta/Elev= 30
       0  731.77    29.2  726.22    48.7  723.03    68.2  720.43    97.5  717.37
   126.7  715.91   165.7  711.42     195  708.77   253.4  708.76   263.2  708.41
   272.9   707.3   282.7  705.36   292.4  703.81   302.2  703.71   311.9  705.06
   331.4  708.95   341.2  709.54   370.2  710.34   437.8  710.94   466.8  711.61
   544.1  715.95   573.1  716.87   582.8   717.7   611.8  721.75   621.4  722.67
   660.1  723.44   679.4  724.36   698.8   725.9   737.4  730.16   776.1  733.18
#Mann= 3 , 0 , 0
       0     .06       0   282.7    .045       0   311.9     .06       0
Bank Sta=282.7,311.9
XS Rating Curve= 0 ,0
Exp/Cntr=0.3,0.1

Type RM Length L Ch R = 1 ,28859.4 ,455.4,469.6,482.8
XS GIS Cut Line= 2
     1838219.975       670571.08     1839183.517      670018.996
#Sta/Elev= 30
       0  759.98    19.6  752.93    29.5  750.12    68.8  742.29    98.3  734.14
   108.1   732.9   147.4  731.92   176.9  729.53   186.7  728.14     226  720.45
   235.9   719.2   265.3  717.68   324.3  710.28     344  709.69   481.5  708.84
   707.6  708.82   717.4  708.64   732.8  706.27   746.9  703.96   756.7  704.56
   766.5  707.39   786.2  714.87   864.8  735.01   923.8  751.15   982.7  766.57
   992.6  770.22  1002.4  774.67  1041.7  793.54  1071.2  808.85  1110.5  830.31
#Mann= 3 , 0 , 0
       0     .06       0   732.8    .045       0   766.5     .08       0
Bank Sta=732.8,766.5
XS Rating Curve= 0 ,0
Exp/Cntr=0.3,0.1

Type RM Length L Ch R = 1 ,28389.8 ,84,83.6,287.1
XS GIS Cut Line= 5
     1838601.083      670750.392     1838880.395       670645.65
     1838969.134      670612.191      1839283.36      670626.739
     1839514.665      670561.275
#Sta/Elev= 30
       0  721.41    19.2  719.37    28.9  718.92   125.1   717.3   192.4  715.08
   221.3  713.39   288.7  711.71   355.2  708.24   393.1  707.54   422.6  708.47
   432.5  708.13   447.7  704.72   452.1  703.71     462  702.94   471.8  703.34
   481.6   704.3   520.9  707.67   589.7   711.2   599.6   712.7   609.4  714.88
   648.7  724.53   668.4  727.76     688  729.96   707.7  731.22   851.9   744.4
   871.2  746.63   890.4  749.34     900  751.35   928.9  758.69   948.1  762.55
#Mann= 3 , 0 , 0
       0     .06       0   447.7    .045       0   481.6     .06       0
Bank Sta=447.7,481.6
XS Rating Curve= 0 ,0
Exp/Cntr=0.3,0.1

Type RM Length L Ch R = 1 ,28306.2 ,339.9,333.9,123.8
XS GIS Cut Line= 5
     1838617.837      670829.435     1838897.149      670724.693
     1838985.888      670691.234     1839300.114      670705.782
     1839531.419      670640.318
#Sta/Elev= 30
       0  723.11     9.6     723    19.2  722.22    28.9  720.21    38.5  718.71
    48.1  718.18   182.8  715.76   355.2  710.29   374.2  709.21   393.1  707.51
   412.8  706.47   452.1  702.76   471.4  702.28   481.6  702.76   501.3   704.6
   511.1  705.06   609.4  706.84   629.1  706.87   638.9  707.17   648.7  708.08
   658.6   709.7   678.2   713.7     688  715.14   726.9  718.94   784.6  726.47
   832.7  733.38   871.2  735.65   890.4  737.63   938.5  745.11   948.1  747.05
#Mann= 3 , 0 , 0
       0     .06       0   452.1    .045       0   481.6     .06       0
Bank Sta=452.1,481.6
XS Rating Curve= 0 ,0
Exp/Cntr=0.3,0.1

Type RM Length L Ch R = 1 ,27972.3 ,669.7,668.9,668.3
XS GIS Cut Line= 4
      1838516.85      671206.496     1838721.379      670968.066
     1839375.786      670764.669     1839563.046      670676.399
#Sta/Elev= 30
       0  821.27    39.3   814.3    49.1  810.66    58.9  803.69    98.2     768
     108  759.97   117.8     755   127.6   752.4   206.2   735.5   245.4  728.71
     265  726.74   304.3  724.74   323.9  720.04   333.7  719.02   480.6   715.1
   588.2  711.41   744.9  707.96   813.4  707.37   901.5  708.18   911.3  707.12
   930.9  702.63   940.7  702.09   950.5  703.08   956.3   704.5   979.8  712.05
   999.4  716.47  1065.3   726.6  1168.8  736.94  1187.6  739.74  1206.4  743.66
#Mann= 3 , 0 , 0
       0     .06       0   930.9    .045       0   956.3     .07       0
Bank Sta=930.9,956.3
XS Rating Curve= 0 ,0
Exp/Cntr=0.3,0.1

Type RM Length L Ch R = 1 ,27303.3 ,802.9,795.1,802.8
XS GIS Cut Line= 3
     1838787.177      671621.741     1839709.052      671343.095
     1839951.239      671426.428
#Sta/Elev= 30
       0  805.65    19.6  795.67    29.5  789.61    68.8  762.61    78.6  757.14
   196.5  721.96     226  717.69   245.7   711.8   255.5  710.09   314.5  706.19
   353.8  704.79   422.6  704.71   501.2  707.12   540.5   707.4   668.2  705.13
   746.9  705.73   766.5  702.01   776.4  701.13   786.2  701.18     796  702.73
   815.7  706.44   884.4  712.62   943.4  727.98    1020  749.88  1067.4   767.2
  1095.9   779.5  1152.8     809  1171.8  817.17  1181.2  819.48  1219.2  821.73
#Mann= 3 , 0 , 0
       0     .06       0   766.5    .045       0     796     .08       0
Bank Sta=766.5,796
XS Rating Curve= 0 ,0
Exp/Cntr=0.3,0.1

Type RM Length L Ch R = 1 ,26508.2 ,1243.2,1263.5,1267.7
XS GIS Cut Line= 3
     1838757.301      671982.972      1839675.27      672147.035
     1840011.208      672096.253
#Sta/Elev= 30
       0  853.13     9.8  848.55    29.4  842.67    88.3  832.76     108   826.8
   137.4   811.9   196.3  769.27   225.8  751.33   333.7  720.35   353.4  716.17
   382.8  713.58   441.7  705.12   520.2  704.23   559.5   701.4   569.3  701.05
   590.5  702.34   657.7  713.65   726.4  734.09   755.8  740.43   804.9  745.78
   903.1  753.55   932.5  760.33   942.2  760.78   961.6  756.03   971.3  755.46
     981  758.34  1107.2  821.37  1165.5  842.36  1223.7  854.61  1272.3   873.4
#Mann= 3 , 0 , 0
       0     .06       0   559.5    .045       0   590.5     .06       0
Bank Sta=559.5,590.5
XS Rating Curve= 0 ,0
Exp/Cntr=0.3,0.1
